--- 15203_ras.prj (project) ---

Proj Title=15203
Current Plan=p01
Default Exp/Contr=0.3,0.1
English Units
Geom File=g01
Flow File=f01
Plan File=p01
Y Axis Title=Elevation
X Axis Title(PF)=Main Channel Distance
X Axis Title(XS)=Station
BEGIN DESCRIPTION:
RFD model 15203 exported to HEC-RAS
END DESCRIPTION:

--- 15203_ras.p01 (plan) ---

Plan Title=Plan 01
Program Version=4.10
Short Identifier=Plan 01
Geom File=g01
Flow File=f01
Subcritical Flow
Calc Critical at every XS
Secant Critical Depth

--- 15203_ras.f01 (steady flow) ---

Flow Title=Flow 01
Program Version=5.01
Number of Profiles= 6
Profile Names=10yr,25yr,50yr,100yr,100plus,500yr
River Rch & RM=15203,37,13916.41
 1024.64 1678.05 2303.63 2885.19 4212.37 5783.61
River Rch & RM=15203,37,13672.59
 1029.79 1686.63 2315.57 2900.28 4234.41 5810.22
River Rch & RM=15203,37,13428.78
 1569.97    2577 3544.33 4443.69 6487.79 8395.88
River Rch & RM=15203,37,13184.96
 1575.78 2586.71 3557.85 4460.82  6512.8 8424.35
River Rch & RM=15203,37,12941.15
 1581.58 2596.41 3571.37 4477.93 6537.78 8452.78
River Rch & RM=15203,37,12697.33
 1590.04 2610.57 3591.09 4502.91 6574.25 8494.26
River Rch & RM=15203,37,12453.51
 1595.14  2619.1 3602.99 4517.99 6596.27 8519.33
River Rch & RM=15203,37, 12209.7
 1602.89 2632.08 3621.08 4540.92 6629.75 8557.43
River Rch & RM=15203,37,11965.88
 1608.86 2642.07 3635.02 4558.59 6655.54 8586.77
River Rch & RM=15203,37,11722.07
 1614.82 2652.06 3648.95 4576.25 6681.32 8616.07
River Rch & RM=15203,37,11478.25
 1619.21 2659.42 3659.22 4589.28 6700.35 8637.75
River Rch & RM=15203,37,11234.44
 1623.59 2666.78 3669.49 4602.31 6719.37 8659.41
River Rch & RM=15203,37,10715.32
 1631.47 2679.99 3687.94 4625.73 6753.56 8698.35
River Rch & RM=15203,37,10568.92
 1633.21 2682.93 3692.04 4630.93 6761.15 8706.99
River Rch & RM=15203,37,10237.96
 1636.93 2689.16 3700.74 4641.98 6777.28 8725.34
River Rch & RM=15203,37,9864.279
 1642.17 2697.95 3713.02 4657.56 6800.04 8751.23
River Rch & RM=15203,37,9490.599
 1647.18 2706.37 3724.78 4672.48 6821.83 8776.01
River Rch & RM=15203,37,9144.035
 2355.13 3892.02 5378.59 6768.65 9882.2312146.19
River Rch & RM=15203,37,8993.551
 2390.75 3951.88 5462.29 6874.9510037.4312313.48
River Rch & RM=15203,37,8504.094
 2411.41 3986.62 5510.86 6936.65 10127.512410.42
River Rch & RM=15203,37,7995.881
 2449.46 4050.56 5600.28  7050.210293.2912588.48
River Rch & RM=15203,37,7815.174
 2473.41 4090.83 5656.59 7121.7210397.7112700.42
River Rch & RM=15203,37,7659.848
 2475.01 4093.51 5660.34 7126.4810404.6712707.87
River Rch & RM=15203,37,7497.642
 2475.81 4094.85 5662.22 7128.8610408.14 12711.6
River Rch & RM=15203,37,7045.841
 2502.88 4140.37 5725.88 7209.7210526.1912837.96
River Rch & RM=15203,37,6594.039
 2506.66 4146.73 5734.76    722110542.6712855.57
River Rch & RM=15203,37,6142.238
 2515.24 4161.12 5754.89 7246.5510579.97 12895.4
River Rch & RM=15203,37,5781.946
 2524.79 4177.18 5777.34 7275.0510621.57 12939.8
River Rch & RM=15203,37,5684.458
 2525.39 4178.18 5778.74 7276.8310624.1712942.58
River Rch & RM=15203,37,5044.849
 2607.98 4316.98 5972.83  7523.310984.0213325.83
River Rch & RM=15203,37,4870.682
 2609.57 4319.64 5976.54 7528.0210990.9113333.14
River Rch & RM=15203,37,4452.518
 2644.31 4378.01 6058.14 7631.6111142.1513493.56
Boundary for River Rch & Prof#=15203,37,1
Up Type= 0
Dn Type= 2
Boundary for River Rch & Prof#=15203,37,2
Up Type= 0
Dn Type= 2
Boundary for River Rch & Prof#=15203,37,2
Up Type= 0
Dn Type= 2
Boundary for River Rch & Prof#=15203,37,2
Up Type= 0
Dn Type= 2
Boundary for River Rch & Prof#=15203,37,2
Up Type= 0
Dn Type= 2
Boundary for River Rch & Prof#=15203,37,2
Up Type= 0
Dn Type= 2

--- 15203_ras.g01 (geometry) ---

Geom Title=15203
Program Version=4.10

River Reach=15203,37
Reach XY= 30
743926.269239535851176.448043176744060.376034319851149.504315466
744268.709367633851221.118898779744593.145131528 851684.44355154
744765.671173215851669.252579346745157.381242663852038.176190495
745429.733673185852088.089384899745634.811798185852392.993898779
745599.655548215852549.894940495745719.447214872852647.551190451
745702.520131558852790.780357137745815.801381588852836.353273794
745696.009714842852965.259523839745699.915964872853134.530357137
745766.322214872853157.967857122746007.207631528853075.936607122
746200.604019463853625.856652945746835.224122226854073.346545607
    749059.18265 854680.98551099749268.383995175854890.186876461
749425.502099663855491.749303699749616.474242091855641.922793403
750472.377046168855557.721664131750979.321360409855588.971590713
 751966.84883523856036.050177738752125.703001857856155.841844454
752297.578001916856418.862677723752386.119668543856689.696011052
752610.078001916857752.196011052 752929.59043479858791.901242375

Type RM Length L Ch R = 1 ,13916.41,243.815500,243.815500,243.815500
XS GIS Cut Line= 6
743623.722820417  852103.5226766743822.053587654851738.492995969
743930.622155587851446.886145882743946.174928331851302.618148264
743913.718019853850840.950391766744072.705676767850198.001429408
#Sta/Elev= 30
8999.098143.8765 9141.34142.4276 9161.58 139.3459261.593141.61719287.515131.0701
9362.653128.9953 9418.49131.78579470.401131.70299495.299123.84239549.471122.7859
 9570.97119.81939666.323118.16099768.928119.80089779.078118.9569 9799.32112.4593
9929.685107.5691 9960.1392.776869980.58587.585389990.89881.0975310001.2277.53193
10021.7583.8056410042.2886.0309710062.6395.2729810072.7697.0144410143.13 98.1246
10163.16100.891510526.37105.854810557.08107.846110742.79106.980911000.91114.4382
#Mann= 3 , 0 , 0
8999.098   0.063       08999.098   0.063       011000.91   0.063       0
#XS Ineff= 2 , 0
       0                               0
Bank Sta=8999.098,11000.91
Exp/Cntr=0.3,0.1

Type RM Length L Ch R = 1 ,13672.59,243.815400,243.815400,243.815400
XS GIS Cut Line= 6
743722.714472363852065.405179254743938.349802646851692.164641207
744079.938518825851404.157171615 744149.07255688851228.806933782
744297.414025995850775.796013175744512.434647419850232.417267379
#Sta/Elev= 30
8999.056140.19839034.468141.10419081.054138.09419162.581140.80679174.228139.7977
9197.521129.62169277.823127.38769323.692129.97289381.028129.71889403.962122.2743
9472.011119.78869550.861121.6724 9573.39118.07789662.114114.5937 9771.87116.2702
  9804.3108.11839847.539107.59799870.747104.78159911.719106.40979954.15594.29897
9975.13485.938029985.46184.185359995.77276.1620510006.0977.2016310035.8993.35731
 10047.595.6508210141.9995.0160610237.0198.3967710438.81101.090511000.9796.97939
#Mann= 3 , 0 , 0
8999.056    0.04       08999.056    0.04       011000.97    0.04       0
#XS Ineff= 2 , 0
       0                               0
Bank Sta=8999.056,11000.97
Exp/Cntr=0.3,0.1

Type RM Length L Ch R = 1 ,13428.78,243.815400,243.815400,243.815400
XS GIS Cut Line= 6
743759.751117497852120.479633643744109.403363453851588.054429617
744324.199035932 851353.62300521 744570.44954334851048.823095198
744700.349165039850845.431619581744900.492317146850484.381848935
#Sta/Elev= 30
8999.075141.14399100.612136.84719194.091138.60439219.396128.99599290.667125.8046
9397.573128.44559421.329121.55859456.965 119.3459578.098121.8887 9594.73121.1584
9615.213114.11579798.671 113.623 9812.27111.92289827.199104.36269952.503100.2243
9965.45693.254219978.23980.9917210002.3774.0747510039.8281.3874910079.92105.7769
10106.65114.636910200.22116.014710238.86 121.66110411.52 124.012 10529.9132.8158
10678.15136.619510784.12145.408310829.61144.468110852.36136.656211000.92134.4381
#Mann= 3 , 0 , 0
8999.075    0.06       08999.075    0.06       011000.92    0.06       0
#XS Ineff= 2 , 0
       0                               0
Bank Sta=8999.075,11000.92
Exp/Cntr=0.3,0.1

Type RM Length L Ch R = 1 ,13184.96,243.815400,243.815400,243.815400
XS GIS Cut Line= 6
743809.273620993 852236.76689169744215.007254697851704.363779936
744349.773292501851591.597009941744576.250900303851462.325273894
744690.713253941851352.653777047745107.234387326850746.727724567
#Sta/Elev= 30
8999.104136.74289164.848134.36819251.421 136.9729258.509136.5027 9286.05 126.388
9320.021126.87599394.478121.79399432.181123.8246 9453.35 118.4119534.339121.5479
9573.425120.55219595.074113.42639624.704111.16219682.801108.96259789.707111.3062
9822.235101.32789932.56797.809079966.38783.0864710000.2271.4933610011.5774.97432
10034.2795.8206910057.07113.2874 10179.2112.803510211.96139.353910248.35145.9124
10318.79148.020210743.43148.532410767.19146.952510790.76142.1294 11000.9134.0712
#Mann= 3 , 0 , 0
8999.104    0.08       08999.104    0.08       0 11000.9    0.08       0
#XS Ineff= 2 , 0
       0                               0
Bank Sta=8999.104,11000.9
Exp/Cntr=0.3,0.1

Type RM Length L Ch R = 1 ,12941.15,243.815500,243.815500,243.815500
XS GIS Cut Line= 6
744103.078736654 852504.45645829 744564.46245296 851934.16241615
744631.501971428851785.968740392744628.828133094 851634.19403684
 744663.60201163851539.964982113745135.485488299 850833.29401936
#Sta/Elev= 30
8999.127122.84829017.283128.39549064.697133.3512 9117.73131.02299169.586133.4318
9210.538129.71669310.004131.28249316.477130.7094 9329.48121.66689342.484117.2099
 9433.51116.70689523.301108.9244 9626.78111.14819648.377 103.6389755.51695.07596
  9789.885.757069968.22583.8130610008.8672.3109410039.1578.5738310069.56 95.2759
10090.52109.745210101.26112.798410226.48111.289310238.41115.654510267.67137.5981
10302.35145.526210360.22147.973810761.01148.577410944.47134.903111000.83132.9029
#Mann= 3 , 0 , 0
8999.127  0.0617       08999.127  0.0617       011000.83  0.0617       0
#XS Ineff= 2 , 0
       0                               0
Bank Sta=8999.127,11000.83
Exp/Cntr=0.3,0.1

Type RM Length L Ch R = 1 ,12697.33,243.815400,243.815400,243.815400
XS GIS Cut Line= 6
744237.820998722852524.847857257744501.442965422852232.182361207
744656.783412612852035.346123161744866.753343629851709.555052609
745152.086396303851293.955492747745410.150970468 850906.63744573
#Sta/Elev= 30
8999.047133.0618 9053.96131.65419107.545133.92549148.309129.05359189.073131.7333
9246.941130.75629262.082127.49599282.663115.50829398.579 112.6779453.926106.7469
9524.907106.41239569.106100.36079607.53386.843149711.752 87.05569752.99780.80262
9966.88879.754569978.51278.138779990.09771.0893710001.6668.9872510013.3672.67122
10049.1896.1850910063.34102.651910207.62106.532810231.82114.076910363.11132.9004
10425.41144.240310582.38145.454210811.34129.661710973.66 123.08811000.98119.0999
#Mann= 3 , 0 , 0
8999.047  0.0616       08999.047  0.0616       011000.98  0.0616       0
#XS Ineff= 2 , 0
       0                               0
Bank Sta=8999.047,11000.98
Exp/Cntr=0.3,0.1

Type RM Length L Ch R = 1 ,12453.51,243.815400,243.815400,243.815400
XS GIS Cut Line= 6
744334.611862648852625.583012763744587.830385742852369.440598373
744880.499610819852047.691364276745141.027350357851778.992191015
745244.677286246851641.304332003 745620.85418052 851098.94077198
#Sta/Elev= 30
8999.019131.33399098.609133.17859183.502128.3026 9312.06131.97239340.781129.3158
9355.142122.33449406.242 121.6329447.213116.29729516.572114.03699561.466106.8016
9636.483 106.6669651.255104.02239666.219 94.55939756.00892.264069770.901 86.3978
9815.04579.202979970.74980.114389981.43678.024799998.787 68.238110013.0469.83751
 10027.380.6725310084.8683.5504610099.7991.3514110256.33108.947610341.48136.6003
10394.12 142.48610591.98140.898210738.02126.7034 10955.6117.353411000.96107.1013
#Mann= 3 , 0 , 0
8999.019  0.0656       08999.019  0.0656       011000.96  0.0656       0
#XS Ineff= 2 , 0
       0                               0
Bank Sta=8999.019,11000.96
Exp/Cntr=0.3,0.1

Type RM Length L Ch R = 1 , 12209.7,243.815400,243.815400,243.815400
XS GIS Cut Line= 6
744508.125137022852773.400749265744911.738209155852430.117547583
745085.488160966 852249.64725544745207.019751184852060.930368227
 745382.97662539851713.814611389745730.730387373851216.558564413
#Sta/Elev= 30
8999.048125.05389105.205122.32059138.801124.34069182.804122.92239230.335128.5733
9353.522128.11819374.175120.76599413.941118.55479440.453113.50399560.762110.2225
9672.602101.08649693.38395.383589759.78993.961759810.46990.117279846.55579.45417
9883.35175.730289976.47276.30421 9999.74 66.746910033.5276.6383910044.7582.74291
10209.1191.9717110254.0897.5544410397.78118.697510428.38124.782110452.21135.4637
10464.12137.914410499.96 139.67410584.73 139.76510699.85126.422911000.95 112.612
#Mann= 3 , 0 , 0
8999.048   0.075       08999.048   0.075       011000.95   0.075       0
#XS Ineff= 2 , 0
       0                               0
Bank Sta=8999.048,11000.95
Exp/Cntr=0.3,0.1

Type RM Length L Ch R = 1 ,11965.88,243.815500,243.815500,243.815500
XS GIS Cut Line= 6
744704.724297979852760.102655606745136.668444346852443.546422902
745270.934176406852323.135513575 745332.78494719 852244.34750899
 745407.63924719852110.916268192746049.561619964851302.588215869
#Sta/Elev= 30
8999.138117.4449 9049.32116.41079086.698118.66389124.076113.34689358.387107.8238
9669.67987.655119698.23784.007869739.11571.486639752.05270.519389976.32172.61414
9995.40865.7814310011.3969.6908610027.1880.9721510066.9396.97442 10253.4125.1253
10367.18125.854910417.96129.2628 10469.5127.180910624.15114.203810662.81114.5201
10692.51109.6104 10765.9 109.57410803.49104.619310830.34104.131210856.1192.00582
10866.9191.6042910882.7691.3518610933.43108.5688 10959.2111.205411000.97110.2399
#Mann= 3 , 0 , 0
8999.138   0.063       08999.138   0.063       011000.97   0.063       0
#XS Ineff= 2 , 0
       0                               0
Bank Sta=8999.138,11000.97
Exp/Cntr=0.3,0.1

Type RM Length L Ch R = 1 ,11722.07,243.815400,243.815400,243.815400
XS GIS Cut Line= 6
744712.788242789852811.429193815745087.433599712852558.168726633
745526.302195288 852312.91709027745738.266463314852167.742316374
 746016.38994114851937.647566871746323.218054727851638.659804841
#Sta/Elev= 30
8999.039111.5181 9062.04114.36269113.922111.26069221.795110.74289290.782106.0763
9389.088106.47179710.55685.074589752.87476.152249784.374 72.76299884.72670.60487
9976.59771.4018710000.33 62.884110059.1989.1535210109.74103.099610163.83104.5939
10219.81117.902810244.88120.934410314.64121.201210471.02107.722310605.81101.5834
10649.93102.257310677.3596.8223110749.1591.7160810804.73 90.592910837.0880.93885
10875.7292.7323610907.52106.791510932.52110.317710975.11110.629611000.97113.5346
#Mann= 3 , 0 , 0
8999.039  0.0693       08999.039  0.0693       011000.97  0.0693       0
#XS Ineff= 2 , 0
       0                               0
Bank Sta=8999.039,11000.97
Exp/Cntr=0.3,0.1

Type RM Length L Ch R = 1 ,11478.25,243.815400,243.815400,243.815400
XS GIS Cut Line= 6
744706.992754437852884.640462438 745291.25577375852545.745795973
745482.418272719852496.608857739745679.803257082852509.523982664
745820.614649315852455.586580089746452.977118803852007.195994477
#Sta/Elev= 30
8999.132109.83939045.606110.65039082.289107.81689118.882110.22979332.099104.6757
9355.609101.90739466.721101.22319626.20689.480629743.59983.997849785.17873.27376
9916.67170.952119926.67366.691739956.82870.618089977.12170.1444110007.5663.79387
10067.9480.5313610251.6699.7752310297.03115.495810320.21120.071610378.44120.5607
10497.08106.238610632.3799.8309210744.9590.3466110860.4988.2252610873.4984.37098
 10886.576.5818510894.8176.2031310910.4581.9314310938.51101.294411000.89104.1661
#Mann= 3 , 0 , 0
8999.132  0.0637       08999.132  0.0637       011000.89  0.0637       0
#XS Ineff= 2 , 0
       0                               0
Bank Sta=8999.132,11000.89
Exp/Cntr=0.3,0.1

Type RM Length L Ch R = 1 ,11234.44,519.118200,519.118200,519.118200
XS GIS Cut Line= 6
744994.293731828852922.789983734745148.906703055852844.110586882
745315.760185093852781.164010644745658.247120798852686.393784478
745775.121370345852681.245438561746041.537879378852528.003580227
#Sta/Elev= 30
9232.48897.907039401.704  96.382 9455.6993.226579520.32987.174989551.98987.63782
9666.82782.682279687.49779.551019832.30766.511029863.54968.632099873.96367.39806
9894.79168.993869926.03367.693489966.88567.736089976.96666.378989987.02262.75732
9997.07860.7560210007.1661.9739210027.2273.5328610040.1378.0590310097.4682.84455
10113.1585.6944210124.4885.37264 10205.891.1823410256.48 92.325910263.9994.56874
10276.02101.998310299.12111.610910310.87115.052510333.18115.647710365.55114.2784
#Mann= 3 , 0 , 0
9232.488  0.0576       09232.488  0.0576       010365.55  0.0576       0
#XS Ineff= 2 , 0
       0                               0
Bank Sta=9232.488,10365.55
Exp/Cntr=0.3,0.1

Type RM Length L Ch R = 1 ,10715.32,146.402500,146.402500,146.402500
XS GIS Cut Line= 6
745374.223390586853314.845796137745464.651599147853217.085570665
745605.276599088853110.141126232745736.943265804853003.474459545
745854.373821326852912.155015142746172.327543297852693.561831267
#Sta/Elev= 30
9580.22988.840029610.82689.953849702.61889.283449716.84491.425559738.96391.77408
9749.88490.89475 9764.0988.369079789.21687.827159826.90684.340859852.03280.66419
9898.237 78.14269915.45374.643859928.32373.029169961.78171.878189966.93270.91801
9979.80264.723839992.67259.6670910069.73 68.880510107.7368.02983 10158.469.87059
10203.6566.9235810209.0467.1832810233.3171.4382910245.4572.3319910306.1274.13593
10397.4279.9114910503.3384.9097310560.9684.2377310585.2386.6075810594.1386.42087
#Mann= 3 , 0 , 0
9580.229  0.0687       09580.229  0.0687       010594.13  0.0687       0
#XS Ineff= 2 , 0
       0                10083.34       0
Bank Sta=9580.229,10594.13
Exp/Cntr=0.3,0.1

Type RM Length L Ch R = 3 ,10651.32,,,
BEGIN DESCRIPTION:
END DESCRIPTION:
Bridge Culvert--1,0,-1,-1, 0
Deck Dist Width WeirC Skew NumUp NumDn MinLoCord MaxHiCord MaxSubmerge Is_Ogee
54.828600,36.745300,2.6,0, 60, 60, , , 0.95, 0, 0,0,,
 9671.77 9692.50 9706.51 9734.54 9748.56 9752.83 9762.57 9764.93 9767.49 9775.28
 9787.72 9800.17 9825.05 9837.50 9849.94 9856.53 9864.45 9951.38 9951.3810009.45
10009.4510051.6710088.9610126.2510138.6810161.6710184.0610206.4410217.6410228.83
10240.0210273.6010284.8010295.9910307.1810318.3810329.5710340.7710352.9410363.15
10375.2010385.5410397.4610407.9310419.1210430.3110442.2010465.9910513.9210525.44
10532.4010537.3310569.3710587.8510596.7810608.6810644.3510668.1310680.0210683.94
   89.99   89.52   89.65   89.17   88.51   88.77   90.67   90.59   90.35   88.71
   87.26   85.96   84.14   82.84   81.85   81.54   80.91   75.14   75.14   71.43
   71.43   68.84   67.61   66.96   67.15   67.13   67.57   68.21   68.75   68.97
   69.50   70.55   71.25   71.50   72.21   72.59   73.29   73.64   74.38   74.70
   75.39   75.72   76.40   76.66   77.29   77.64   78.27   79.20   80.60   81.15
   81.17   81.47   82.50   82.89   83.35   83.32   85.17   85.93   86.50   86.34
 -910.01 -910.48 -910.35 -910.83 -911.49 -911.23 -909.33 -909.41 -909.65 -911.29
 -912.74 -914.04 -915.86 -917.16 -918.15 -918.46 -919.09 -924.86   71.64   67.93
 -928.57 -931.16 -932.39 -933.04 -932.85 -932.87 -932.43 -931.79 -931.25 -931.03
 -930.50 -929.45 -928.75 -928.50 -927.79 -927.41 -926.71 -926.36 -925.62 -925.30
 -924.61 -924.28 -923.60 -923.34 -922.71 -922.36 -921.73 -920.80 -919.40 -918.85
 -918.83 -918.53 -917.50 -917.11 -916.65 -916.68 -914.83 -914.07 -913.50 -913.66
 9671.77 9692.50 9706.51 9734.54 9748.56 9752.83 9762.57 9764.93 9767.49 9775.28
 9787.72 9800.17 9825.05 9837.50 9849.94 9856.53 9864.45 9951.23 9951.2310009.31
10009.3110051.6710088.9610126.2510138.6810161.6710184.0610206.4410217.6410228.83
10240.0210273.6010284.8010295.9910307.1810318.3810329.5710340.7710352.9410363.15
10375.2010385.5410397.4610407.9310419.1210430.3110442.2010465.9910513.9210525.44
10532.4010537.3310569.3710587.8510596.7810608.6810644.3510668.1310680.0210683.94
   89.99   89.52   89.65   89.17   88.51   88.77   90.67   90.59   90.35   88.71
   87.26   85.96   84.14   82.84   81.85   81.54   80.91   75.15   75.15   71.44
   71.44   68.84   67.61   66.96   67.15   67.13   67.57   68.21   68.75   68.97
   69.50   70.55   71.25   71.50   72.21   72.59   73.29   73.64   74.38   74.70
   75.39   75.72   76.40   76.66   77.29   77.64   78.27   79.20   80.60   81.15
   81.17   81.47   82.50   82.89   83.35   83.32   85.17   85.93   86.50   86.34
 -910.01 -910.48 -910.35 -910.83 -911.49 -911.23 -909.33 -909.41 -909.65 -911.29
 -912.74 -914.04 -915.86 -917.16 -918.15 -918.46 -919.09 -924.85   71.65   67.94
 -928.56 -931.16 -932.39 -933.04 -932.85 -932.87 -932.43 -931.79 -931.25 -931.03
 -930.50 -929.45 -928.75 -928.50 -927.79 -927.41 -926.71 -926.36 -925.62 -925.30
 -924.61 -924.28 -923.60 -923.34 -922.71 -922.36 -921.73 -920.80 -919.40 -918.85
 -918.83 -918.53 -917.50 -917.11 -916.65 -916.68 -914.83 -914.07 -913.50 -913.66
BR Coef=-1 , 0 , 0 ,, 0 ,,,0.8,0,1,0,
WSPro=,,,, 1 ,,,, 0 ,,,, 0 ,,,,-1 ,-1 ,-1 , 0 , 0 , 0 , 0 , 0
BC Design=,, 0 ,, 0 ,,,,,,

Type RM Length L Ch R = 1 ,10568.92,330.958000,330.958000,330.958000
XS GIS Cut Line= 5
745475.249775019853411.033239675745824.850627601853085.400294259
 745909.57284981853006.233627588746206.696111619852866.376065031
746280.178825051852820.969293997
#Sta/Elev= 30
9632.294 90.64779754.946 88.49649773.192 89.98469836.94288.181639850.60885.35712
9875.89583.193389891.60679.794569919.911 78.5239 9946.2768.496659963.92665.69339
9978.598 65.7236 9993.2759.8575310007.9457.7019610022.6159.8184710028.27 62.2436
10051.96 63.952410066.6367.1640610082.93 65.406910151.3265.9956810169.2367.37135
10198.5267.5012210232.0169.9219310298.3271.2256910322.8373.8348910386.7476.22565
10408.8578.4112310464.1180.9199910497.2780.6600810541.4882.4212510640.7883.49578
#Mann= 3 , 0 , 0
9632.294  0.0677       09632.294  0.0677       010640.78  0.0677       0
#XS Ineff= 2 , 0
       0                               0
Bank Sta=9632.294,10640.78
Exp/Cntr=0.3,0.1

Type RM Length L Ch R = 1 ,10237.96,373.679500,373.679500,373.679500
XS GIS Cut Line= 6
744402.402037382855007.288908079744972.023426771854338.298233941
745755.754880607853488.507247522745977.240902752853138.164878771
746534.361310601852848.917162001746970.020851612852535.814493909
#Sta/Elev= 30
7499.163105.7518 7541.26 103.8697567.33596.735947721.40488.350488397.20467.62656
8557.47969.038558719.57461.946188993.30861.780179007.06960.162499020.82952.18016
9046.73355.23393 9062.1163.043129119.521 74.63429367.37586.531939580.69482.90089
9646.35778.173069664.66268.235179676.856 67.3816 9783.0663.028379894.74166.74811
9983.32962.435519994.11857.4393110036.8169.0679710320.3768.1640610404.9778.83691
10614.9776.2923910662.2462.4711410716.0585.2285510770.46101.097511115.77110.0332
#Mann= 3 , 0 , 0
7499.163  0.0623       07499.163  0.0623       011115.77  0.0623       0
#XS Ineff= 2 , 0
       09878.905        10164.87       0
Bank Sta=7499.163,11115.77
Exp/Cntr=0.3,0.1

Type RM Length L Ch R = 1 ,9864.279,373.679500,373.679500,373.679500
XS GIS Cut Line= 6
745239.066023278854334.997102064745928.114845824853590.917377791
746058.016599072853504.204745476746589.906589267853241.699805596
746864.845470989853038.336414236747156.667251998852773.729597926
#Sta/Elev= 30
 8749.0966.000458864.25166.503788879.41769.92159  8908.770.244348948.60366.61017
9175.36867.967399364.15761.426489391.12763.586819405.38570.249499479.25378.47062
9569.54879.876739611.18374.978859746.46576.026699916.82770.565999939.09664.71135
9983.30663.676419994.35853.0374810005.3254.5019410026.8362.6635210048.3363.32175
10123.6161.2132910243.6464.5510810368.1362.9051710497.1165.4190510667.0862.33658
10732.7864.0603710818.5474.5794110936.0683.2001810985.0298.4713611250.92111.6751
#Mann= 3 , 0 , 0
 8749.09  0.0787       0 8749.09  0.0787       011250.92  0.0787       0
#XS Ineff= 2 , 0
       09699.329         10422.1       0
Bank Sta=8749.09,11250.92
Exp/Cntr=0.3,0.1

Type RM Length L Ch R = 1 ,9490.599,346.564300,346.564300,346.564300
XS GIS Cut Line= 6
744968.710089394855800.135896499746219.885768439853991.493252605
746452.772012259853599.615756835746551.494032553853492.209264763
747070.613128729853026.568467896747471.810214777852607.094028363
#Sta/Elev= 30
7499.029128.5686 7835.82112.96397969.911115.54658018.671107.09178323.39496.53639
8347.65390.50638 8432.5687.234518565.98689.567478735.53184.19898 8929.8987.31885
9111.81784.433479353.94671.71351    959772.948879780.28267.802819801.62863.87737
9958.74863.755329974.31162.156719985.403 51.443510007.5450.6511210018.5953.82968
10029.7361.8440610466.7260.5828210735.4968.0827910750.4573.8808610880.7186.30074
10894.4493.7040311032.42102.381911391.09105.388711538.49103.179311578.88106.8308
#Mann= 3 , 0 , 0
7499.029  0.0778       07499.029  0.0778       011578.88  0.0778       0
#XS Ineff= 2 , 0
       0 9646.31        10444.01       0
Bank Sta=7499.029,11578.88
Exp/Cntr=0.3,0.1

Type RM Length L Ch R = 1 ,9144.035,150.483500,150.483500,150.483500
XS GIS Cut Line= 6
745449.677016467856090.087794289746609.399238765854031.060016513
746696.899238735853843.560016483 746783.01034981853554.671127602
747088.565905362853138.004460931747537.834123671852612.650495961
#Sta/Elev= 30
7517.596142.72427742.779125.10967812.034 127.1937962.088123.44978077.514113.9229
8366.079105.30268429.285110.20258585.25199.737698677.312100.34058746.35897.39876
8769.37393.489948986.61790.126739157.72678.752089306.02177.451359648.23966.28489
9887.56764.324219965.06559.4552910008.9649.5499510019.9958.7286810031.0359.30906
10190.6457.3530910629.3563.9895510711.2568.3754810760.8588.6827310832.2789.65099
10975.68   99.39 11069.796.9435611362.04103.265411462.5399.50073 11597.2104.4239
#Mann= 3 , 0 , 0
7517.596  0.0773       07517.596  0.0773       0 11597.2  0.0773       0
#XS Ineff= 2 , 0
       0                10444.59       0
Bank Sta=7517.596,11597.2
Exp/Cntr=0.3,0.1

Type RM Length L Ch R = 3 ,9079.481,,,
BEGIN DESCRIPTION:
END DESCRIPTION:
Bridge Culvert--1,0,-1,-1, 0
Deck Dist Width WeirC Skew NumUp NumDn MinLoCord MaxHiCord MaxSubmerge Is_Ogee
45.058100,60.367300,2.6,0, 31, 31, , , 0.95, 0, 0,0,,
 9650.97 9658.17 9669.70 9704.27 9715.80 9738.85 9773.42 9796.47 9807.68 9818.69
 9840.70 9862.71 9884.72 9895.72 9906.73 9979.82 9979.8210020.1810020.1810042.60
10057.0810069.0210079.7310085.1410090.4310101.1310111.8410197.4010218.6810239.96
10316.91
   66.08   66.07   66.21   66.21   65.91   64.82   63.35   62.81   62.44   62.22
   61.48   60.88   60.43   60.32   60.09   59.37   59.37   58.98   58.98   58.77
   57.78   57.47   56.92   56.72   56.66   56.75   56.62   57.68   57.75   57.95
   58.96
 -933.92 -933.93 -933.79 -933.79 -934.09 -935.18 -936.65 -937.19 -937.56 -937.78
 -938.52 -939.12 -939.57 -939.68 -939.91 -940.63   56.37   55.98 -941.02 -941.23
 -942.22 -942.53 -943.08 -943.28 -943.34 -943.25 -943.38 -942.32 -942.25 -942.05
 -941.04
 9650.97 9658.17 9669.70 9704.27 9715.80 9738.85 9773.42 9796.47 9807.68 9818.69
 9840.70 9862.71 9884.72 9895.72 9906.73 9979.82 9979.8210020.1810020.1810042.60
10057.0810069.0210079.7310085.1410090.4310101.1310111.8410197.4010218.6810239.96
10316.91
   66.08   66.07   66.21   66.21   65.91   64.82   63.35   62.81   62.44   62.22
   61.48   60.88   60.43   60.32   60.09   59.37   59.37   58.98   58.98   58.77
   57.78   57.47   56.92   56.72   56.66   56.75   56.62   57.68   57.75   57.95
   58.96
 -933.92 -933.93 -933.79 -933.79 -934.09 -935.18 -936.65 -937.19 -937.56 -937.78
 -938.52 -939.12 -939.57 -939.68 -939.91 -940.63   56.37   55.98 -941.02 -941.23
 -942.22 -942.53 -943.08 -943.28 -943.34 -943.25 -943.38 -942.32 -942.25 -942.05
 -941.04
BR Coef=-1 , 0 , 0 ,, 0 ,,,0.8,0,1,0,
WSPro=,,,, 1 ,,,, 0 ,,,, 0 ,,,,-1 ,-1 ,-1 , 0 , 0 , 0 , 0 , 0
BC Design=,, 0 ,, 0 ,,,,,,

Type RM Length L Ch R = 1 ,8993.551,489.457500,489.457500,489.457500
XS GIS Cut Line= 6
745544.121460915856154.671127617746706.621460885854154.671127602
746849.677016467853832.448905379746871.899238735853671.337794289
747029.538127631853426.893349841747663.533210695852623.229131997
#Sta/Elev= 30
7544.961143.97887765.603136.77717880.011127.10317984.497126.71848157.608117.1086
 8284.84118.88868442.184108.29138661.078105.69748700.87796.366248805.33592.28038
 8979.4792.47026  9025.1 82.49499098.86678.738679117.63280.904389152.33276.33079
9417.25776.166119476.95668.667829591.86168.967669936.16759.710629969.708 58.3496
9991.31548.4784110013.1648.53942   1002458.5214610508.5263.0833510666.9180.78038
10908.3586.8163410965.0893.5576511175.2193.9330311314.9999.4104311688.1596.60765
#Mann= 3 , 0 , 0
7544.961   0.075       07544.961   0.075       011688.15   0.075       0
#XS Ineff= 2 , 0
       0                10471.88       0
Bank Sta=7544.961,11688.15
Exp/Cntr=0.3,0.1

Type RM Length L Ch R = 1 ,8504.094,508.212700,508.212700,508.212700
XS GIS Cut Line= 6
746180.699437288856374.909924119746893.124937387855062.291866306
747136.913628463854476.322308349747397.446358381853709.366524931
747606.393032378853349.189069574748092.111827397852659.297629432
#Sta/Elev= 30
7555.273139.42477636.924132.4285 8031.51121.54978095.902104.70988177.338111.7547
8443.006112.22518465.721120.82218521.989121.35298544.495120.25398578.254108.5821
8735.764107.82798891.59695.686399406.70571.209389594.21972.71618 9696.3958.67295
9969.107 53.339610000.04 43.698810020.6346.8542810030.9253.9661410144.3261.93677
10249.5159.12175 10346.566.0601510512.5565.9915710603.1969.7181810626.2575.65503
10738.5674.8048610823.5387.0647811336.0488.6917611456.1396.9352211756.72103.8639
#Mann= 3 , 0 , 0
7555.273   0.075       07555.273   0.075       011756.72   0.075       0
#XS Ineff= 2 , 0
       0                10461.77       0
Bank Sta=7555.273,11756.72
Exp/Cntr=0.3,0.1

Type RM Length L Ch R = 1 ,7995.881,180.707700,180.707700,180.707700
XS GIS Cut Line= 6
746760.891437322856605.328253374747342.297809243855467.122311994
747549.390076697854922.092901021747929.029413313 853630.30406104
748104.124746174853237.695864573748364.892101318852770.024920836
#Sta/Elev= 30
7499.033137.63687568.312140.97667831.526138.92198243.862125.91818294.263116.0749
8372.392117.74458494.138105.32668604.599101.18758714.496103.79088877.502 91.7701
9039.38589.395129060.84384.013949326.27381.641589420.81773.863739535.89274.50593
 9639.7864.594659970.85556.374379981.17943.216919991.50441.4967210012.1641.50014
10022.4953.2463810032.8355.1884310084.5157.1768410448.5362.3540510554.0873.41284
11093.7582.12642   1111986.3021311231.1686.05288 11459.299.3942311673.77105.1283
#Mann= 3 , 0 , 0
7499.033  0.0661       07499.033  0.0661       011673.77  0.0661       0
#XS Ineff= 2 , 0
       0                10463.52       0
Bank Sta=7499.033,11673.77
Exp/Cntr=0.3,0.1

Type RM Length L Ch R = 1 ,7815.174,155.325500,155.325500,155.325500
XS GIS Cut Line= 6
746955.927016467856609.532238752747380.927016467855767.865572065
747768.427016526854832.448905408748118.427016497853540.782238737
 748333.01034984852999.115572065748444.901239663852836.282488525
#Sta/Elev= 30
7545.436138.92367987.413132.15318054.629125.86718386.428118.25678408.613 113.085
8631.818110.20828923.426 95.88239054.879 85.30969157.73782.742149248.41984.78977
9346.10975.946539454.65277.092559487.21671.666839549.93668.347769705.14565.77904
9974.17455.454739984.52141.7030510005.2241.1161610015.5641.9791810025.9154.60152
 10263.958.1283610533.5867.5932610689.3577.0669410813.9680.0630410845.3384.08672
11017.4378.67526 11221.884.6813711442.91 95.286511487.39100.709411619.31 103.057
#Mann= 3 , 0 , 0
7545.436  0.0749       07545.436  0.0749       011619.31  0.0749       0
#XS Ineff= 2 , 0
       0                10461.24       0
Bank Sta=7545.436,11619.31
Exp/Cntr=0.3,0.1

Type RM Length L Ch R = 3 ,7739.455,,,
BEGIN DESCRIPTION:
END DESCRIPTION:
Bridge Culvert--1,0,-1,-1, 0
Deck Dist Width WeirC Skew NumUp NumDn MinLoCord MaxHiCord MaxSubmerge Is_Ogee
48.135250,59.055000,2.6,0, 60, 60, , , 0.95, 0, 0,0,,
 7549.09 7573.16 7595.36 7650.85 7684.15 7706.73 7728.55 7750.75 7772.95 7784.05
 7798.92 7861.74 7883.94 7906.14 7928.34 7939.43 7972.73 7994.93 8017.13 8072.63
 8172.52 8194.72 8239.11 8272.41 8350.11 8383.41 8394.50 8405.60 8438.90 8461.10
 8505.50 8560.99 8594.29 8605.39 8616.49 8805.18 8848.36 8869.94 8945.49 8956.29
 8967.08 8973.61 8977.87 8988.67 9031.84 9085.80 9159.66 9301.66 9639.72 9900.70
 9983.60 9983.6010016.4010016.4010117.3710245.1910410.9910566.1010741.9010904.75
  137.74  137.76  136.75  137.71  135.59  134.82  132.80  132.37  132.27  133.32
  133.28  132.27  131.20  130.91  131.61  131.03  131.16  130.45  127.75  124.30
  123.58  122.49  122.17  120.86  116.22  115.19  113.50  112.76  113.42  113.19
  111.79  108.78  109.04  106.57  102.27  102.12  100.95  101.50   98.72   98.88
   96.91   94.07   91.45   89.99   87.24   85.52   82.13   77.52   64.67   55.96
   55.08   55.08   54.86   54.86   54.17   56.13   60.04   65.97   74.07   76.84
 -862.26 -862.24 -863.25 -862.29 -864.41 -865.18 -867.20 -867.63 -867.73 -866.68
 -866.72 -867.73 -868.80 -869.09 -868.39 -868.97 -868.84 -869.55 -872.25 -875.70
 -876.42 -877.51 -877.83 -879.14 -883.78 -884.81 -886.50 -887.24 -886.58 -886.81
 -888.21 -891.22 -890.96 -893.43 -897.73 -897.88 -899.05 -898.50 -901.28 -901.12
 -903.09 -905.93 -908.55 -910.01 -912.76 -914.48 -917.87 -922.48 -935.33 -944.04
 -944.92   52.58   52.36 -945.14 -945.83 -943.87 -939.96 -934.03 -925.93 -923.16
 7549.09 7573.16 7595.36 7650.85 7684.15 7706.73 7728.55 7750.75 7772.95 7784.05
 7798.92 7861.74 7883.94 7906.14 7928.34 7939.43 7972.73 7994.93 8017.13 8072.63
 8172.52 8194.72 8239.11 8272.41 8350.11 8383.41 8394.50 8405.60 8438.90 8461.10
 8505.50 8560.99 8594.29 8605.39 8616.49 8805.18 8848.36 8869.94 8945.49 8956.29
 8967.08 8973.61 8977.87 8988.67 9031.84 9085.80 9159.66 9301.66 9639.72 9900.70
 9983.60 9983.6010016.4010016.4010117.3710245.1910410.9910566.1010741.9010904.75
  137.74  137.76  136.75  137.71  135.59  134.82  132.80  132.37  132.27  133.32
  133.28  132.27  131.20  130.91  131.61  131.03  131.16  130.45  127.75  124.30
  123.58  122.49  122.17  120.86  116.22  115.19  113.50  112.76  113.42  113.19
  111.79  108.78  109.04  106.57  102.27  102.12  100.95  101.50   98.72   98.88
   96.91   94.07   91.45   89.99   87.24   85.52   82.13   77.52   64.67   55.96
   55.08   55.08   54.86   54.86   54.17   56.13   60.04   65.97   74.07   76.84
 -862.26 -862.24 -863.25 -862.29 -864.41 -865.18 -867.20 -867.63 -867.73 -866.68
 -866.72 -867.73 -868.80 -869.09 -868.39 -868.97 -868.84 -869.55 -872.25 -875.70
 -876.42 -877.51 -877.83 -879.14 -883.78 -884.81 -886.50 -887.24 -886.58 -886.81
 -888.21 -891.22 -890.96 -893.43 -897.73 -897.88 -899.05 -898.50 -901.28 -901.12
 -903.09 -905.93 -908.55 -910.01 -912.76 -914.48 -917.87 -922.48 -935.33 -944.04
 -944.92   52.58   52.36 -945.14 -945.83 -943.87 -939.96 -934.03 -925.93 -923.16
BR Coef=-1 , 0 , 0 ,, 0 ,,,0.8,0,1,0,
WSPro=,,,, 1 ,,,, 0 ,,,, 0 ,,,,-1 ,-1 ,-1 , 0 , 0 , 0 , 0 , 0
BC Design=,, 0 ,, 0 ,,,,,,

Type RM Length L Ch R = 1 ,7659.848,162.206100,162.206100,162.206100
XS GIS Cut Line= 6
747050.024238706856677.587794304747677.802016526855399.810016498
747888.913127631854884.532238737748018.600627571854488.525294289
748118.427016497854139.393349826748560.985150665852932.414477333
#Sta/Elev= 30
7501.539 137.1187916.666131.28288039.225124.83498128.359124.8672 8170.48115.5508
8284.343117.94048574.028106.22678585.169102.44078918.849 98.45058952.01596.26998
8984.435 88.39659427.51274.988199471.72973.123379513.12666.593629776.19162.90974
9975.22454.804299985.62541.434799994.78241.0964910016.8342.9316310027.2353.76724
10120.8358.0331210266.5557.0380410468.71 61.372410745.3577.0881411032.6277.69669
11149.6684.5163711181.5890.10922 11266.7 88.999911394.3897.0806511547.8299.31882
#Mann= 3 , 0 , 0
7501.539  0.0714       07501.539  0.0714       011547.82  0.0714       0
#XS Ineff= 2 , 0
       0                10464.48       0
Bank Sta=7501.539,11547.82
Exp/Cntr=0.3,0.1

Type RM Length L Ch R = 1 ,7497.642,451.801300,451.801300,451.801300
XS GIS Cut Line= 6
747185.767052501  856706.3504695747607.267461896855936.889352679
747938.567469597855245.433858559 748095.37868908854816.912904009
748403.202770561853762.396763682748716.947310239853061.570640713
#Sta/Elev= 30
7499.035135.51527981.815123.42188004.599120.71638031.028109.94958129.514107.0611
8242.721107.17558524.698 96.89198558.205100.36488803.43798.374998891.83490.40682
8980.06789.892229001.90182.290259034.65380.242219056.487 74.47429601.82660.17954
    992458.696949965.44356.944669975.804  52.2379986.16540.8526410017.2541.73647
10027.6251.6669210037.9853.67795 10089.854.2765210110.5357.9145510547.9261.93363
10664.1469.7488710932.2271.06808 11124.485.8757911261.41 91.278911467.1293.15964
#Mann= 3 , 0 , 0
7499.035  0.0688       07499.035  0.0688       011467.12  0.0688       0
#XS Ineff= 2 , 0
       0                10463.41       0
Bank Sta=7499.035,11467.12
Exp/Cntr=0.3,0.1

Type RM Length L Ch R = 1 ,7045.841,451.801400,451.801400,451.801400
XS GIS Cut Line= 6
747479.765615211856750.429876498748438.843714271855092.410227678
748562.608544135854806.473279781748957.126116975853650.373087382
749268.972985558 853027.47492893749699.080046323852289.009979079
#Sta/Elev= 30
7499.044132.7746 7760.75128.71997830.376119.81398269.869113.6749 8397.09107.8146
8443.35396.217698580.47491.168278790.86195.138248871.996  75.833 9115.8864.93868
9968.25956.118829999.35940.6019210020.0644.2119910030.4155.5692110459.1260.32497
11291.8787.11605 11489.273.7904911658.7775.0104511700.1965.2084912085.1557.38946
12120.4742.7546712132.0949.0223612144.3273.9960212190.1977.03376 12271.779.33365
12319.6671.1703912353.5952.1522712376.9847.6001612447.1752.9636612500.9765.28806
#Mann= 3 , 0 , 0
7499.044   0.075       07499.044   0.075       012500.97   0.075       0
#XS Ineff= 2 , 0
       0                10613.08       0
Bank Sta=7499.044,12500.97
Exp/Cntr=0.3,0.1

Type RM Length L Ch R = 1 ,6594.039,451.801300,451.801300,451.801300
XS GIS Cut Line= 6
747665.255810166856751.399715717748320.343121371855686.504607041
748523.410826358855403.166623855748902.738870538854937.030324141
749010.023556029854787.289637334750343.782430176852535.200590502
#Sta/Elev= 30
7499.054129.1893  7681.2122.92487902.477122.52748655.50496.818298715.35980.71619
8775.09972.363599058.50169.262069083.37862.366299172.19959.635849967.38653.51741
9990.31639.61014    999939.4677710013.2639.5891410036.1753.3019110151.6857.01244
10669.4653.75543 11316.765.5796511420.6956.9637711559.3654.8078811570.9144.55593
11582.57 41.384511594.0241.7223311617.1354.8093511640.2458.7595611778.9158.01914
11802.0267.4934511921.8569.1026411980.9581.6284212103.6777.5995512500.9886.82091
#Mann= 3 , 0 , 0
7499.054  0.0816       07499.054  0.0816       012500.98  0.0816       0
#XS Ineff= 2 , 0
       0                10493.45       0
Bank Sta=7499.054,12500.98
Exp/Cntr=0.3,0.1

Type RM Length L Ch R = 1 ,6142.238,360.291800,360.291800,360.291800
XS GIS Cut Line= 6
747674.290168687856847.339075929748679.153260618855356.417507441
749001.962077429855127.795749189749552.977317821854973.698965766
749792.922576687854777.616897808750788.244864486853143.016229694
#Sta/Elev= 30
7461.755130.62727906.347123.43267992.107115.3299  8687.397.005658739.644  80.683
8794.786 73.00069128.65667.882939168.45261.443869310.49357.76354 9966.5851.81768
9976.72150.938879986.86337.7144110017.2940.05389 10037.651.1949510332.79 54.0355
11372.7548.2536111406.2236.0715211426.4236.28101 11441.849.8833911464.8251.76267
11579.9151.8248711628.4443.8218311709.2571.6857411867.6374.6509811890.6479.48086
12088.8979.4003512147.8692.9004812343.9994.2936112414.31104.860812463.53103.9614
#Mann= 3 , 0 , 0
7461.755   0.077       07461.755   0.077       012463.53   0.077       0
#XS Ineff= 2 , 0
       0                10664.09       0
Bank Sta=7461.755,12463.53
Exp/Cntr=0.3,0.1

Type RM Length L Ch R = 1 ,5781.946,97.487700,97.487700,97.487700
XS GIS Cut Line= 6
748507.894609094856816.129460946749012.061275721855661.962794289
749270.394609153855411.962794259749527.339053541855380.018349826
749705.909990132855252.043049589750852.802016497853392.518349826
#Sta/Elev= 30
8265.17499.607848604.69395.49983 8724.7399.013138932.06689.390669008.45391.66404
 9084.84 82.87359257.19980.48306 9282.1872.449749379.47666.96272 9570.4965.38379
9635.32354.357819949.24950.100589989.55736.1919510009.7136.2171110029.8749.41447
10911.2251.7020811561.0847.9920511572.6638.9360611595.8235.24756 11604.636.42441
11624.4452.4077711796.5751.2638211870.2774.96452 11985.473.4320912072.9475.78723
12109.7982.2180212294.9681.8264612330.6891.1581112449.7489.9727112547.9598.86609
#Mann= 3 , 0 , 0
8265.174  0.0793       08265.174  0.0793       012547.95  0.0793       0
#XS Ineff= 2 , 0
       0                10901.01       0
Bank Sta=8265.174,12547.95
Exp/Cntr=0.3,0.1

Type RM Length L Ch R = 3 ,5731.319,,,
BEGIN DESCRIPTION:
END DESCRIPTION:
Bridge Culvert--1,0,-1,-1, 0
Deck Dist Width WeirC Skew NumUp NumDn MinLoCord MaxHiCord MaxSubmerge Is_Ogee
16.243850,65.000000,2.6,0, 31, 31, , , 0.95, 0, 0,0,,
 9841.24 9846.24 9849.31 9859.51 9869.71 9879.91 9890.11 9896.88 9900.31 9910.51
 9920.72 9930.92 9935.15 9978.21 9978.2110013.2110013.2110041.2910043.1310048.82
10053.3310063.5310073.7310083.9310094.1310099.4710104.3310114.5310124.7310134.93
10141.95
   50.29   50.21   50.17   50.23   50.23   49.95   49.88   49.86   49.84   49.74
   49.74   49.71   49.65   49.43   49.43   49.26   49.26   49.12   49.12   49.13
   49.11   49.07   49.11   49.01   48.79   48.75   48.74   48.69   48.68   48.62
   48.47
 -949.71 -949.79 -949.83 -949.77 -949.77 -950.05 -950.12 -950.14 -950.16 -950.26
 -950.26 -950.29 -950.35 -950.57   46.93   46.76 -950.74 -950.88 -950.88 -950.87
 -950.89 -950.93 -950.89 -950.99 -951.21 -951.25 -951.26 -951.31 -951.32 -951.38
 -951.53
 9841.24 9846.24 9849.31 9859.51 9869.71 9879.91 9890.11 9896.88 9900.31 9910.51
 9920.72 9930.92 9935.15 9969.96 9969.9610004.9610004.9610041.2910043.1310048.82
10053.3310063.5310073.7310083.9310094.1310099.4710104.3310114.5310124.7310134.93
10141.95
   50.29   50.21   50.17   50.23   50.23   49.95   49.88   49.86   49.84   49.74
   49.74   49.71   49.65   49.47   49.47   49.30   49.30   49.12   49.12   49.13
   49.11   49.07   49.11   49.01   48.79   48.75   48.74   48.69   48.68   48.62
   48.47
 -949.71 -949.79 -949.83 -949.77 -949.77 -950.05 -950.12 -950.14 -950.16 -950.26
 -950.26 -950.29 -950.35 -950.53   46.97   46.80 -950.70 -950.88 -950.88 -950.87
 -950.89 -950.93 -950.89 -950.99 -951.21 -951.25 -951.26 -951.31 -951.32 -951.38
 -951.53
BR Coef=-1 , 0 , 0 ,, 0 ,,,0.8,0,1,0,
WSPro=,,,, 1 ,,,, 0 ,,,, 0 ,,,,-1 ,-1 ,-1 , 0 , 0 , 0 , 0 , 0
BC Design=,, 0 ,, 0 ,,,,,,

Type RM Length L Ch R = 1 ,5684.458,639.610000,639.610000,639.610000
XS GIS Cut Line= 6
748556.852942377856848.073905393 749102.68627575855723.073905393
749319.352942377855506.407238707 749540.18627575855464.740572035
749779.769609094855300.157238707750919.005720198853434.879460916
#Sta/Elev= 30
8337.563100.62398663.31193.597168785.57596.405638985.64287.942729074.56189.74998
9107.90682.99234 9163.4881.268169295.47681.563479319.08975.389819585.84661.20821
9961.20550.086589971.38149.288329981.55838.0232210001.9135.3530210022.2638.01788
10042.6249.3831610662.4351.3962811554.5947.5547211581.4734.9028711601.9635.78082
 11618.853.9924911791.4552.3965811826.9859.7703311862.5174.2460612104.1275.68134
12141.4582.8998812324.3883.9569712549.3992.3507212570.7799.2471412596.9199.03069
#Mann= 3 , 0 , 0
8337.563  0.0924       08337.563  0.0924       012596.91  0.0924       0
#XS Ineff= 2 , 0
       0                10942.39       0
Bank Sta=8337.563,12596.91
Exp/Cntr=0.3,0.1

Type RM Length L Ch R = 1 ,5044.849,174.166300,174.166300,174.166300
XS GIS Cut Line= 6
749065.880720198856974.462794274749754.769609094856418.907238707
750010.325164646856096.685016483749965.880720168 855388.35168317
750045.741831303855162.657238722751267.964053512853218.212794289
#Sta/Elev= 30
8222.22980.48671 8587.7675.37377 8901.9778.970999097.51576.717779201.55170.05498
9507.86968.956689541.001 64.17759655.23265.953849736.28455.835659857.56256.94945
9887.88247.696529968.734  45.512 9978.8442.476689988.94732.7006210009.16  32.106
10019.2735.5863810029.3745.4188910575.7549.6318311210.5345.9628111230.6734.19287
11270.9446.7723611292.6662.44888 11472.359.0642911546.1371.5286211741.99 72.2692
11814.6180.69857 12179.883.7532212271.9787.3053612297.8693.2668712778.3192.78247
#Mann= 3 , 0 , 0
8222.229  0.0924       08222.229  0.0924       012778.31  0.0924       0
#XS Ineff= 2 , 0
       0                 10719.4       0
Bank Sta=8222.229,12778.31
Exp/Cntr=0.3,0.1

Type RM Length L Ch R = 3 ,4937.451,,,
BEGIN DESCRIPTION:
END DESCRIPTION:
Bridge Culvert--1,0,-1,-1, 0
Deck Dist Width WeirC Skew NumUp NumDn MinLoCord MaxHiCord MaxSubmerge Is_Ogee
65.757750,42.650800,2.6,0, 35, 35, , , 0.95, 0, 0,0,,
 9517.50 9521.37 9532.13 9542.88 9553.63 9575.14 9579.41 9585.89 9596.64 9633.84
 9656.08 9681.03 9711.30 9721.40 9731.49 9741.58 9751.67 9761.77 9771.86 9781.95
 9812.23 9822.32 9862.69 9882.88 9903.06 9930.33 9983.60 9983.6010016.4010016.40
10069.9810074.6410086.6210094.8210105.93
   64.05   63.49   62.83   63.10   62.82   62.44   62.46   62.23   61.34   58.73
   58.14   56.98   55.87   55.37   54.98   54.68   54.65   54.92   54.44   53.72
   51.94   51.40   49.52   48.23   47.24   46.29   45.81   45.81   45.51   45.51
   45.03   45.21   45.31   45.51   45.91
 -935.95 -936.51 -937.17 -936.90 -937.18 -937.56 -937.54 -937.77 -938.66 -941.27
 -941.86 -943.02 -944.13 -944.63 -945.02 -945.32 -945.35 -945.08 -945.56 -946.28
 -948.06 -948.60 -950.48 -951.77 -952.76 -953.71 -954.19   43.31   43.01 -954.49
 -954.97 -954.79 -954.69 -954.49 -954.09
 9517.50 9521.37 9532.13 9542.88 9553.63 9575.14 9579.41 9585.89 9596.64 9633.84
 9656.08 9681.03 9711.30 9721.40 9731.49 9741.58 9751.67 9761.77 9771.86 9781.95
 9812.23 9822.32 9862.69 9882.88 9903.06 9930.33 9983.60 9983.6010016.4010016.40
10069.9810074.6410086.6210094.8210105.93
   64.05   63.49   62.83   63.10   62.82   62.44   62.46   62.23   61.34   58.73
   58.14   56.98   55.87   55.37   54.98   54.68   54.65   54.92   54.44   53.72
   51.94   51.40   49.52   48.23   47.24   46.29   45.81   45.81   45.51   45.51
   45.03   45.21   45.31   45.51   45.91
 -935.95 -936.51 -937.17 -936.90 -937.18 -937.56 -937.54 -937.77 -938.66 -941.27
 -941.86 -943.02 -944.13 -944.63 -945.02 -945.32 -945.35 -945.08 -945.56 -946.28
 -948.06 -948.60 -950.48 -951.77 -952.76 -953.71 -954.19   43.31   43.01 -954.49
 -954.97 -954.79 -954.69 -954.49 -954.09
BR Coef=-1 , 0 , 0 ,, 0 ,,,0.8,0,1,0,
WSPro=,,,, 1 ,,,, 0 ,,,, 0 ,,,,-1 ,-1 ,-1 , 0 , 0 , 0 , 0 , 0
BC Design=,, 0 ,, 0 ,,,,,,
